--- LONGRN1.prj (project) ---

Proj Title=LONGRN1
Current Plan=p01
Default Exp/Contr=0,0
English Units
Geom File=g01
Flow File=f01
Plan File=p01
BEGIN DESCRIPTION:
Stream Name: Long Run 1
Flood Zone: Approximate
Pendleton County, West Virginia
HEC-RAS Version: 5.0.7
Hydrology Method:
Regression
Model Notes:
NA
END DESCRIPTION:
DSS File=dss
DSS Export Rating Curves= 0
DSS Export Rating Curve Sorted= 0
DSS Export Volume Flow Curves= 0
DXF OffsetX= 0
DXF OffsetY= 0
DXF ScaleX= 0
DXF ScaleY= 0

--- LONGRN1.p01 (plan) ---

Plan Title=Floodplain
Program Version=5.07
Short Identifier=Floodplain
Geom File=g01
Flow File=f01
Subcritical Flow
K Sum by GR= 0
Std Step Tol= 0.01
Critical Tol= 0.01
Num of Std Step Trials= 20
Max Error Tol= 0.3
Flow Tol Ratio= 0.001
Split Flow NTrial= 30
Split Flow Tol= 0.02
Split Flow Ratio= 0.02
Log Output Level= 0
Friction Slope Method= 1
Unsteady Friction Slope Method= 2
Unsteady Bridges Friction Slope Method= 1
Parabolic Critical Depth
Global Vel Dist= 0 , 0 , 0
Global Log Level= 0
CheckData=False
Encroach Param=-1 ,0,0, 0
Computation Interval=0.1SEC
Output Interval=1MIN
Instantaneous Interval=Max Profile
Mapping Interval=1HOUR
Computation Time Step Use Courant=        0
Computation Time Step Use Time Series=    0
Computation Time Step Count To Double=0
Computation Time Step Max Doubling=0
Computation Time Step Max Halving=0
Computation Time Step Residence Courant=0
Run HTab= 0
Run UNet= 0
Run Sediment= 0
Run PostProcess= 0
Run WQNet= 0
Run RASMapper= 0
UNET Theta= 0
UNET Theta Warmup= 0
UNET ZTol= 0
UNET ZSATol= 0
UNET MxIter= 0
UNET Max Iter WO Improvement= 0
UNET MaxInSteps= 0
UNET DtIC= 0
UNET DtMin= 0
UNET MaxCRTS= 0
UNET WFStab= 0
UNET SFStab= 0
UNET WFX= 1
UNET SFX= 1
UNET 1D Methodology=Finite Difference
UNET DSS MLevel= 1
UNET Pardiso=0
UNET DZMax Abort= 0
UNET Use Existing IB Tables= 0
UNET Froude Reduction=False
UNET Froude Limit= 0
UNET Froude Power= 0
UNET D1 Cores= 0
UNET D2 Coriolis=0
UNET D2 Cores= 0
UNET D2 Theta= 1
UNET D2 Theta Warmup= 1
UNET D2 Z Tol= 0.01
UNET D2 Volume Tol= 0.01
UNET D2 Max Iterations= 20
UNET D2 Equation= 0
UNET D2 RampUpFraction=0.1
UNET D2 TimeSlices= 1
UNET D2 BCVolumeCheck=0
UNET D1D2 MaxIter= 0
UNET D1D2 ZTol=0.01
UNET D1D2 QTol=0.1
UNET D1D2 MinQTol=1
DSS File=dss
Write IC File= 0
Write IC File at Fixed DateTime=0
Write IC File at Sim End=0
Echo Input=False
Echo Parameters=False
Echo Output=False
Write Detailed= 0
HDF Write Warmup=0
HDF Write Time Slices=0
HDF Flush=0
HDF Face Node Velocities=0
HDF Compression= 1
HDF Chunk Size= 1
HDF Spatial Parts= 1
HDF Use Max Rows=0
HDF Fixed Rows= 1
Calibration Method= 0
Calibration Iterations= 20
Calibration Max Change=0.05
Calibration Tolerance=0.2
Calibration Maximum=1.5
Calibration Minimum=0.5
Calibration Optimization Method= 1
WQ AD Non Conservative
WQ ULTIMATE=-1
WQ Max Comp Step=1HOUR
WQ Output Interval=15MIN
WQ Output Selected Increments= 0
WQ Output face flow=0
WQ Output face velocity=0
WQ Output face area=0
WQ Output face dispersion=0
WQ Output cell volume=0
WQ Output cell surface area=0
WQ Output cell continuity=0
WQ Output cumulative cell continuity=0
WQ Output face conc=0
WQ Output face dconc_dx=0
WQ Output face courant=0
WQ Output face peclet=0
WQ Output face adv mass=0
WQ Output face disp mass=0
WQ Output cell mass=0
WQ Output cell source sink temp=0
WQ Output nsm pathways=0
WQ Output nsm derived pathways=0
WQ Output MaxMinRange=-1
WQ Daily Max Min Mean=-1
WQ Daily Range=0
WQ Daily Time=0
WQ Create Restart=0
WQ Fixed Restart=0
WQ System Summary=0
WQ Write To DSS=0
WQ Use Fixed Temperature=0
Sorting and Armoring Iterations= 10
XS Update Threshold= 0.02
Bed Roughness Predictor= 0
Hydraulics Update Threshold= 0.02
Energy Slope Method= 1
Volume Change Method= 1
Sediment Retention Method= 0
XS Weighting Method= 0
Number of US Weighted Cross Sections= 1
Number of DS Weighted Cross Sections= 1
Upstream XS Weight=0
Main XS Weight=1
Downstream XS Weight=0
Number of DS XS's Weighted with US Boundary= 1
Upstream Boundary Weight= 1
Weight of XSs Associated with US Boundary= 0
Number of US XS's Weighted with DS Boundary= 1
Downstream Boundary Weight= 0.5
Weight of XSs Associated with DS Boundary= 0.5
Percentile Method= 0
Sediment Output Level= 3
Mass or Volume Output= 0
Output Increment Type= 1
Profile and TS Output Increment= 1
XS Output Flag= 0
XS Output Increment= 10
Write Gradation File= 0
Read Gradation Hotstart= 0
Write HDF5 File= 1
Write Binary Output= 1
Write DSS Sediment File= 0
SV Curve= 0
Specific Gage Flag= 0

--- LONGRN1.f01 (steady flow) ---

Flow Title=Flows
Program Version=5.07
Number of Profiles= 6
Profile Names=P100yr,P10yr,P25yr,P50yr,P500yr,P101yr
River Rch & RM=LONGRN1,Main            ,14776
     572     267     378     472     838     696
River Rch & RM=LONGRN1,Main            ,12492
     665     310     439     549     976     809
River Rch & RM=LONGRN1,Main            ,10997
     772     360     509     637    1135     939
River Rch & RM=LONGRN1,Main            ,8404
    1036     480     681     853    1527    1260
River Rch & RM=LONGRN1,Main            ,4626
    1156     535     760     952    1707    1407
Boundary for River Rch & Prof#=LONGRN1,Main            , 1
Up Type= 0
Dn Type= 3
Dn Slope=0.01788
Boundary for River Rch & Prof#=LONGRN1,Main            , 2
Up Type= 0
Dn Type= 3
Dn Slope=0.01788
Boundary for River Rch & Prof#=LONGRN1,Main            , 3
Up Type= 0
Dn Type= 3
Dn Slope=0.01788
Boundary for River Rch & Prof#=LONGRN1,Main            , 4
Up Type= 0
Dn Type= 3
Dn Slope=0.01788
Boundary for River Rch & Prof#=LONGRN1,Main            , 5
Up Type= 0
Dn Type= 3
Dn Slope=0.01788
Boundary for River Rch & Prof#=LONGRN1,Main            , 6
Up Type= 0
Dn Type= 3
Dn Slope=0.01788
DSS Import GetInterval= 0
DSS Import GetPeak= 0
DSS Import FillOption= 0

--- LONGRN1.g01 (geometry) ---

Geom Title=Geometry
Program Version=5.07

River Reach=LONGRN1         ,Main
Reach XY= 30
2420031.98500004553983.337000012     2420217.472554030.657000005
2420374.90100002554478.6009999962420513.63500002554602.686000004
     2420374.463554832.731999993     2420348.792555115.810000002
2420759.01200002555531.0559999942420823.14600003555698.216000021
     2420996.854555734.8900000162421194.50100002555983.206000015
2421448.59599999556031.8390000022421542.61500004556174.070000008
     2421853.516556310.1050000192422647.72999999557217.179000005
2423677.70300001      557560.9122424105.23000002557583.653999999
2424503.32600003557371.5630000082425211.47700003557445.311000004
2426143.20900002556872.4800000042426646.13600004556825.093999997
2426860.49100003556961.4960000072427423.74900001556597.528999999
2428026.53299999556515.8830000162428164.14600003556408.943000004
2428524.46100003556643.6589999942429275.20700002556708.137999997
     2430527.616556188.5269999952430869.82800001      556212.809
2430993.47000003555863.7389999932431195.82231012555813.788434058

Type RM Length L Ch R = 1 ,14776   ,156.1,156.1,156.1
XS GIS Cut Line= 3
2419941.59270592 554490.582751372420057.25506732554062.772712471
     2419967.254      553677.984
#Sta/Elev= 30
       0 2769.45    65.9 2758.22    93.7 2751.37   119.8 2742.43   186.1 2716.82
   214.3  2707.1   240.4 2699.85   273.1 2692.24   289.7 2683.38   326.9 2656.98
   357.8 2636.66   389.1 2622.06   400.2  2619.9   426.3 2617.47     480    2615
   495.9 2611.64   525.1 2601.16   529.2 2600.46   537.4 2601.23   549.7 2603.87
   590.8 2605.39     599 2606.56   607.3 2609.37   627.8 2619.71   636.4 2623.03
   681.2 2630.94   762.9 2653.57   800.3 2662.02   812.6 2663.74   838.3 2670.37
#Mann= 3 ,-1 , 0
       0      .1       0   525.1    .045       0   537.4      .1       0
Bank Sta=525.1,537.4
XS Rating Curve= 0 ,0
Exp/Cntr=0.3,0.1

Type RM Length L Ch R = 1 ,14620   ,161.5,162.1,167.7
XS GIS Cut Line= 3
2419988.32098392554501.8619908882420120.75815518554076.330932801
     2420391.968      553771.004
#Sta/Elev= 30
       0 2764.36    19.8 2760.89    42.1 2754.37    78.5 2742.15   162.2  2709.3
   191.6 2699.82   229.6 2690.66     267 2678.78   325.4 2653.36   384.2 2623.27
     401 2616.75   411.6 2614.87   463.7    2610   481.9 2607.07     506 2599.38
     526 2598.37   537.3 2598.93     543 2597.42   548.1 2597.07   557.1 2597.46
   562.8 2598.54   568.5  2601.2   591.1 2617.64     608 2625.12   622.3 2634.26
   661.5 2656.12   704.2 2684.25   736.3  2702.8   811.2 2742.97   854.1 2762.84
#Mann= 3 ,-1 , 0
       0      .1       0     543    .045       0   557.1      .1       0
Bank Sta=543,557.1
XS Rating Curve= 0 ,0
Exp/Cntr=0.3,0.1

Type RM Length L Ch R = 1 ,14458   ,139,139.9,140.6
XS GIS Cut Line= 3
2419992.25872757554503.7287050282420183.27476065554163.511859022
2420535.99378524 553895.00648632
#Sta/Elev= 30
       0 2763.71    10.1 2762.09    17.5 2760.07    37.6 2753.28   100.9 2726.69
   152.3 2703.06   205.4 2683.13   271.5 2654.56   299.1 2643.55   312.4 2638.95
   347.6 2624.11   386.2 2610.12   403.1  2601.5   417.5 2592.34   422.2 2591.32
   428.7 2592.52   437.3 2594.35   442.4 2594.59   468.7 2593.54   483.5 2598.28
   508.7  2602.1   522.8 2607.29   537.2 2614.18     558 2626.01   602.8 2655.67
   648.6 2680.24   658.5 2687.35   663.5 2690.08   734.4 2725.62   833.5 2772.53
#Mann= 3 ,-1 , 0
       0      .1       0   417.5    .045       0   428.7      .1       0
Bank Sta=417.5,428.7
XS Rating Curve= 0 ,0
Exp/Cntr=0.3,0.1

Type RM Length L Ch R = 1 ,14318   ,145.7,146.6,146.9
XS GIS Cut Line= 3
2419997.85886999554507.1882089212420254.58698961554279.321263941
     2420584.708      554047.119
#Sta/Elev= 30
       0 2762.99    10.8 2760.22    30.7 2752.85    57.4 2740.47   149.6 2694.61
   223.3 2652.96   271.3 2627.96   296.9  2615.6   325.3 2604.49   350.8 2590.69
   357.8 2588.88   385.3 2588.93   394.9 2586.94   399.7 2586.19   408.3 2586.86
   414.4 2587.67   429.1 2586.82     434 2587.77   438.9 2589.59   453.5 2597.77
   462.1  2600.1     480 2602.83   505.9 2610.06   552.5 2628.38   570.9 2636.99
     592 2648.65     610 2661.85     635 2678.16   663.8 2693.52   746.9 2735.37
#Mann= 3 ,-1 , 0
       0      .1       0   394.9    .045       0   408.3      .1       0
Bank Sta=394.9,408.3
XS Rating Curve= 0 ,0
Exp/Cntr=0.3,0.1

Type RM Length L Ch R = 1 ,14172   ,146,146.1,145.9
XS GIS Cut Line= 3
2420042.82991608554559.9787280532420312.83807759554387.455366124
2420677.22657049554187.807750261
#Sta/Elev= 30
       0 2759.06    35.6 2744.25    83.7 2720.51   100.7  2711.1     140 2687.63
   184.6 2658.04   225.4 2634.14     257 2616.74   315.6 2592.64   338.6 2584.33
   350.2 2581.65   356.8 2581.27   361.4 2581.67   370.5 2584.19   375.1 2584.72
   393.3 2584.01   411.6 2584.82   420.7 2587.38   429.8 2591.73   438.9 2594.66
   493.7 2602.65   507.3 2605.85   520.8 2609.98   543.8 2620.02   562.9 2626.88
   594.8  2643.3   607.7 2650.59   630.1 2665.83   657.8 2682.94   735.9 2716.76
#Mann= 3 ,-1 , 0
       0      .1       0   350.2    .045       0   361.4      .1       0
Bank Sta=350.2,361.4
XS Rating Curve= 0 ,0
Exp/Cntr=0.3,0.1

Type RM Length L Ch R = 1 ,14026   ,154.1,154.1,154.6
XS GIS Cut Line= 3
2420045.17922054 554582.29712042 2420361.9775459554523.093961205
     2420726.434      554302.518
#Sta/Elev= 30
       0 2759.85     7.8 2758.25      24 2752.73    64.7 2734.02    93.2 2718.58
   125.8 2698.36   178.7 2660.38   211.2 2638.49   247.8 2617.24   280.4 2604.46
   292.6 2601.69     318 2593.13   330.3 2587.77   344.8 2578.62   349.92576.559
   353.6 2576.13   364.82576.754   376.9 2578.91   414.4 2578.04   451.8 2585.73
   479.8 2589.59   503.2 2596.31   525.4 2605.11   554.3 2614.34   580.7 2620.38
   606.1 2627.89   654.7 2647.22   685.6 2662.77     732 2677.64   748.3 2683.91
#Mann= 3 ,-1 , 0
       0      .1       0   349.9    .045       0   364.8      .1       0
Bank Sta=349.9,364.8
XS Rating Curve= 0 ,0
Exp/Cntr=0.3,0.1

Type RM Length L Ch R = 1 ,13872   ,136.1,144.2,153.6
XS GIS Cut Line= 3
2420042.69939917554605.1375804452420411.93282785554645.071415309
     2420834.154      554451.458
#Sta/Elev= 30
       0  2754.7    42.4 2748.07    54.4 2743.52    82.6 2729.25   118.8 2707.43
   179.1 2664.35   227.4 2631.92   259.6 2612.78     280 2603.54   303.8 2595.89
   360.2 2581.19   388.7 2578.07   406.8 2574.55   429.5 2572.75   464.7 2573.32
   477.9 2571.36   482.2  2571.1   488.3 2571.42   499.9 2575.62   543.9 2579.58
   575.8 2593.43     612 2615.05   649.5 2641.27   661.3  2646.2   719.9 2687.25
     770 2717.96   781.5  2726.5   794.7 2730.33   803.5    2737   835.9 2754.09
#Mann= 3 ,-1 , 0
       0      .1       0   477.9    .045       0   488.3      .1       0
Bank Sta=477.9,488.3
XS Rating Curve= 0 ,0
Exp/Cntr=0.3,0.1

Type RM Length L Ch R = 1 ,13727   ,152.2,149.6,147.4
XS GIS Cut Line= 3
2420045.30973746554631.2409633312420387.59836358554694.883361857
     2420810.568       554891.47
#Sta/Elev= 30
       0 2744.52    56.5 2732.82    80.9 2724.46    93.1 2718.92   109.1 2709.65
   162.2 2672.25   231.4  2627.7     268 2605.88   297.7 2592.42   324.9    2582
   345.3 2576.68   394.2 2568.89   415.6 2569.53   437.7 2566.89   442.4 2566.52
   448.4 2566.95   459.7 2569.94   469.5 2574.04   521.5 2599.91   571.9 2630.42
   609.7 2654.81   622.9 2664.96   631.7  2666.3   636.1 2668.25   651.9 2680.71
   728.8 2728.06     742  2731.7   762.5 2742.01   781.7 2749.73   814.6 2758.71
#Mann= 3 ,-1 , 0
       0      .1       0   437.7    .045       0   448.4      .1       0
Bank Sta=437.7,448.4
XS Rating Curve= 0 ,0
Exp/Cntr=0.3,0.1

Type RM Length L Ch R = 1 ,13578   ,91.9,89.6,88.6
XS GIS Cut Line= 3
2420027.87750181554718.1817938792420306.98688282554825.785160826
     2420807.853      554937.466
#Sta/Elev= 30
       0  2724.6   115.8 2673.65   180.7 2642.11   232.5 2612.38   258.2 2596.14
   296.8 2576.82   325.6 2565.76   337.9  2564.2   354.2 2564.51   360.62562.735
   366.5 2562.13   371.9 2562.82   395.2  2565.1   419.8 2564.51   423.9    2565
   432.1 2568.69   445.7 2571.34   489.5 2590.83   546.8 2620.14   559.1 2627.88
   575.5 2635.26   606.5 2653.33   624.7 2666.31   641.1 2671.85   653.4 2680.74
     707 2708.03   747.6 2725.63     764 2728.66   784.5 2738.02   812.3 2745.15
#Mann= 3 ,-1 , 0
       0      .1       0   360.6    .045       0   371.9      .1       0
Bank Sta=360.6,371.9
XS Rating Curve= 0 ,0
Exp/Cntr=0.3,0.1

Type RM Length L Ch R = 1 ,13488   ,123.5,120.7,120.9
XS GIS Cut Line= 2
2419992.91762473 554867.69097589     2420813.254      554976.056
#Sta/Elev= 30
       0 2729.42    59.8  2700.4   141.7 2656.68   229.9  2611.4   298.5 2573.49
   318.6 2564.28   330.7 2560.58   350.9  2559.9   379.1 2561.92   399.3 2561.58
   412.6 2560.05   419.2 2559.79   421.5 2560.02   427.5 2561.42   443.7  2569.7
   455.8 2571.21     476 2578.99   512.1 2602.32     523 2608.11   560.7 2625.73
     605  2644.7     630 2658.19   641.4 2666.12   657.5    2671   669.6 2679.07
   698.1 2688.96   734.1 2705.05   786.4 2725.11   798.7 2725.87   827.5 2735.43
#Mann= 3 ,-1 , 0
       0      .1       0   412.6    .045       0   421.5      .1       0
Bank Sta=412.6,421.5
XS Rating Curve= 0 ,0
Exp/Cntr=0.3,0.1

Type RM Length L Ch R = 1 ,13367   ,226.6,221.9,218.3
XS GIS Cut Line= 2
2419976.82047046555005.296483323     2420819.911      555013.766
#Sta/Elev= 30
       0 2706.89    45.1 2695.86      60 2694.06      76 2688.85     156  2647.9
     248 2605.45     256 2600.67     272 2587.44     296 2564.28     304  2558.5
     344 2557.02     352 2555.19     360 2554.62  361.22 2555.17     372 2559.14
     416 2559.94     452 2564.35     468 2568.51     500 2585.33     512 2588.95
     536  2604.6     592 2631.74     616 2646.57     632 2651.38     661 2667.15
     672 2669.56   693.3 2679.02     764 2704.05     828 2723.39   843.1 2723.95
#Mann= 3 ,-1 , 0
       0      .1       0     352    .045       0  361.22      .1       0
Bank Sta=352,361.22
XS Rating Curve= 0 ,0
Exp/Cntr=0.3,0.1

Type RM Length L Ch R = 1 ,13145   ,176,171.9,167.8
XS GIS Cut Line= 3
2419968.84915066555230.1266191142420357.47686621 555232.93818401
2420817.15629369555021.573278826
#Sta/Elev= 30
       0 2680.74      48 2662.45     112 2635.47   147.6 2622.38   310.4 2579.77
   323.9 2574.46   347.9 2568.07   392.3 2562.01   441.52548.724     450 2547.65
   456.62548.497   467.1 2550.55   492.2  2549.2   506.7 2549.63   513.3 2551.39
   533.1 2561.61   543.5 2564.24     564 2572.41   579.7  2580.3   590.4 2587.01
   600.8 2589.27   609.8 2595.65   643.8    2614   692.6 2647.66   712.3 2659.09
   735.6 2667.99   747.9 2669.91   753.2 2672.89   792.9 2687.27   894.6 2722.63
#Mann= 3 ,-1 , 0
       0      .1       0   441.5    .045       0   456.6      .1       0
Bank Sta=441.5,456.6
XS Rating Curve= 0 ,0
Exp/Cntr=0.3,0.1

Type RM Length L Ch R = 1 ,12974   ,153.8,153.8,153.6
XS GIS Cut Line= 3
     2420228.499      555614.0622420580.20910406555282.601234229
2420823.79092567555034.043403373
#Sta/Elev= 30
       0 2631.33    39.3 2618.73    77.3 2604.82   121.3 2591.66   154.3 2589.43
   253.2 2575.58   278.8 2570.05   313.7 2560.71   350.5 2556.27     376 2551.67
   404.3 2541.71   409.9 2541.04   415.12541.833   429.1 2546.29   456.6 2547.12
   471.3 2551.62   528.8 2581.04   540.1 2584.28   550.1 2591.31   586.9 2613.46
   628.5 2642.42   644.7 2652.09   666.9  2662.2   678.9 2663.04   690.1 2669.07
   718.2 2679.75   749.4 2689.27     789 2703.17   820.1 2715.36   831.3 2721.74
#Mann= 3 ,-1 , 0
       0      .1       0   404.3    .045       0   415.1      .1       0
Bank Sta=404.3,415.1
XS Rating Curve= 0 ,0
Exp/Cntr=0.3,0.1

Type RM Length L Ch R = 1 ,12820   ,143.8,144.1,144.9
XS GIS Cut Line= 3
     2420335.792      555727.7112420728.59802411  555352.4951599
     2420893.539      555117.198
#Sta/Elev= 30
       0 2646.15   120.2 2597.69   148.4 2588.28   179.6 2580.65   267.3 2567.43
   287.1 2561.81   311.1 2561.67     338 2556.21   349.3 2555.48   394.6 2541.78
   400.12538.455   406.6 2537.14   415.12538.477   427.3 2541.26   487.7 2537.04
   499.3 2543.16   516.2 2544.86   532.4 2549.56   549.4 2557.88   569.7 2570.22
   589.2  2585.4   607.7  2592.8   636.4 2618.89   654.9 2632.94   672.2 2642.86
   691.8 2651.67   706.4 2654.01   716.2 2658.12   728.3 2659.53   830.6 2700.25
#Mann= 3 ,-1 , 0
       0      .1       0   400.1    .045       0   415.1      .1       0
Bank Sta=400.1,415.1
XS Rating Curve= 0 ,0
Exp/Cntr=0.3,0.1

Type RM Length L Ch R = 1 ,12676   ,183.5,183.4,182.5
XS GIS Cut Line= 3
     2420412.025      555796.1392420852.65602411555438.266005622
2421103.99759663555317.663457214
#Sta/Elev= 30
       0 2640.96   114.3 2592.89   160.7 2586.63   217.8 2572.24   317.1 2553.73
     337 2548.72   371.9  2544.6   387.4 2540.56   402.4 2539.44   430.8 2533.71
   436.5 2532.95   443.52533.619   465.2 2533.87   490.6 2537.63   536.8 2537.45
   553.1 2541.71   579.3 2557.19   616.5 2583.78   638.7 2602.34   660.9 2624.89
   702.2 2651.15   720.2 2657.06   731.9 2665.14   744.1 2668.07   753.1  2674.2
   789.5 2693.13   816.2 2704.49     825 2709.79   837.1 2712.67   846.4 2718.72
#Mann= 3 ,-1 , 0
       0      .1       0   430.8    .045       0   443.5      .1       0
Bank Sta=430.8,443.5
XS Rating Curve= 0 ,0
Exp/Cntr=0.3,0.1

Type RM Length L Ch R = 1 ,12492   ,177.4,175.7,172.1
XS GIS Cut Line= 3
2420518.71948695555937.6357006872420782.98046284555720.011611493
2421157.91224347555365.155721174
#Sta/Elev= 30
       0 2641.06    85.9 2608.43   111.5 2596.25   134.2 2594.35     174 2587.27
   220.3 2574.65   272.1 2557.53   281.9 2556.35   342.3 2540.69   361.6 2539.33
   372.3  2534.6   383.3 2526.34   386.9 2525.67   394.12526.537   403.8 2530.28
   466.1 2527.98   482.4 2530.97   518.6 2531.12   530.3 2534.59   548.5  2544.9
   570.8 2560.21   620.1 2597.91   640.8 2611.88   698.1 2639.18   720.7 2653.43
     732 2655.53   816.9 2706.67   829.4 2710.65   844.5 2721.85   858.6 2730.05
#Mann= 3 ,-1 , 0
       0      .1       0   383.3    .045       0   394.1      .1       0
Bank Sta=383.3,394.1
XS Rating Curve= 0 ,0
Exp/Cntr=0.3,0.1

Type RM Length L Ch R = 1 ,12317   ,112.2,114.1,116
XS GIS Cut Line= 4
2420568.38565809555984.9272695822420931.51958643555809.808700618
2421011.22116352555678.0924182392421265.31405384555449.598670956
#Sta/Elev= 30
       0 2626.65    49.3 2613.05   106.7 2593.29   160.3 2587.08   200.2 2578.78
   281.2 2547.24   316.4 2536.34     329 2534.53   420.8 2531.26   434.7 2529.28
   448.8 2523.07     479 2523.62   493.6  2521.1   500.2 2520.65   505.42521.042
   525.6 2527.22   544.5 2536.29   551.8  2541.2   566.2 2546.49   627.8 2588.34
   663.7  2608.7   702.1 2627.71   730.4 2646.58   747.4 2650.91   755.9 2657.43
   807.3 2686.67   828.1 2701.12   843.7 2706.18     855 2716.75   898.8 2746.93
#Mann= 3 ,-1 , 0
       0      .1       0   493.6    .045       0   505.4      .1       0
Bank Sta=493.6,505.4
XS Rating Curve= 0 ,0
Exp/Cntr=0.3,0.1

Type RM Length L Ch R = 1 ,12202   ,141.8,140.9,140.5
XS GIS Cut Line= 3
2420664.45360787556030.6291450352421017.04310968 555855.17528807
     2421337.186       555501.31
#Sta/Elev= 30
       0 2601.39    53.9    2587   134.4 2575.56   164.2 2567.45   219.2 2547.55
   277.5 2532.16   295.4 2532.26   362.2 2526.07     389 2525.38   405.1 2522.02
   436.3 2520.99   456.2 2517.32   461.8 2516.87   469.1 2517.49   481.7 2518.29
   488.7 2520.67   501.5 2529.55   518.5 2543.56   529.8 2547.59   541.1 2556.85
   603.4 2594.94   658.6 2625.22   679.5  2638.6     694 2642.54   703.3 2650.63
   770.5 2690.76   782.7 2699.64     796 2704.05     815 2719.17     871 2759.16
#Mann= 3 ,-1 , 0
       0      .1       0   456.2    .045       0   469.1      .1       0
Bank Sta=456.2,469.1
XS Rating Curve= 0 ,0
Exp/Cntr=0.3,0.1

Type RM Length L Ch R = 1 ,12062   ,199.6,195.9,191.9
XS GIS Cut Line= 3
2420751.34688107556109.1634033732421084.10557252555981.909641224
     2421423.807       555585.99
#Sta/Elev= 30
       0 2581.19    18.4 2578.06      37 2572.93    55.6 2572.23   142.8 2559.28
   194.2 2548.04   228.4 2536.84   262.7  2530.2   288.4 2526.92   335.5 2525.79
   358.9    2522   387.9 2514.16   433.3 2512.85   439.4 2512.04   448.22512.927
   486.2 2515.24   492.2 2516.69   523.4 2539.96   537.6 2543.86   618.6 2593.33
   670.9  2622.8   682.7 2631.18     695 2635.02   713.4  2648.6   756.4 2672.64
     782 2688.69   792.5 2696.91   807.1 2701.02   818.9 2711.41   877.9 2747.77
#Mann= 3 ,-1 , 0
       0      .1       0   433.3    .045       0   448.2      .1       0
Bank Sta=433.3,448.2
XS Rating Curve= 0 ,0
Exp/Cntr=0.3,0.1

Type RM Length L Ch R = 1 ,11866   ,178.9,181.8,181.8
XS GIS Cut Line= 3
     2421097.458      556377.7862421265.94170631556090.621854966
     2421456.189      555611.225
#Sta/Elev= 30
       0 2595.58    71.8 2587.63   114.8 2579.66   171.2 2560.84   226.7 2546.96
   250.1 2539.06     291 2522.61   305.6 2518.56   337.1 2514.62   358.6 2514.39
   380.1 2510.06   388.7 2506.42   410.2 2508.52  421.45 2507.08   427.4 2506.25
   432.52507.041   439.7 2509.23   453.3 2509.59   470.5 2513.03   473.6 2514.73
   535.5 2563.36   609.1 2608.59   618.4 2615.32   633.8 2619.83     643 2626.75
   681.3 2645.39   758.8 2692.77   771.7 2696.13   784.9 2706.03   848.7 2740.04
#Mann= 3 ,-1 , 0
       0      .1       0  421.45    .045       0   432.5      .1       0
Bank Sta=421.45,432.5
XS Rating Curve= 0 ,0
Exp/Cntr=0.3,0.1

Type RM Length L Ch R = 1 ,11684   ,164.8,165.9,164.3
XS GIS Cut Line= 3
2421227.03686059556439.8256765772421464.08334753556002.789726796
     2421493.492      555628.289
#Sta/Elev= 30
       0 2593.03    92.3 2581.86   142.3 2571.47   192.4 2552.65   255.1 2521.28
   280.3 2513.19   301.6 2510.74   329.5 2509.73   360.7 2505.68   442.6 2503.43
   456.5 2500.55   465.2 2500.09   468.1 2500.45   474.5  2502.3     479 2505.31
   533.3 2547.07   544.5 2557.36   553.5 2569.39   581.5 2589.22   589.5 2593.43
   601.5 2596.81   618.5 2610.02   701.8 2656.54   733.9 2670.98   749.9 2674.81
     760 2679.85   798.1 2694.86   810.1 2697.07   822.2 2703.33   872.8 2724.94
#Mann= 3 ,-1 , 0
       0      .1       0   456.5    .045       0   468.1      .1       0
Bank Sta=456.5,468.1
XS Rating Curve= 0 ,0
Exp/Cntr=0.3,0.1

Type RM Length L Ch R = 1 ,11518   ,86.4,86.4,86.3
XS GIS Cut Line= 4
      2421241.38      556450.4472421504.15821374556220.182929294
2421590.63000429556074.7580369082421601.54513579555727.158836477
#Sta/Elev= 30
       0 2592.78    89.5 2582.15   129.7 2575.72   217.6 2546.27   254.3 2531.13
   308.2 2511.51   353.7 2500.65   374.3 2499.68   383.6 2497.19   397.5    2497
   402.62495.403   411.6  2494.1   417.12495.492   432.4 2501.04   464.6 2503.53
     486 2507.61   509.3 2508.93   522.6 2512.18   534.6 2517.08   550.6 2525.76
   594.2 2552.98   610.6 2560.47   646.6 2583.98   658.6  2584.9   670.6 2594.22
   714.5 2613.39   742.7 2622.48   818.7 2651.49   830.7 2653.69   866.4 2667.29
#Mann= 3 ,-1 , 0
       0      .1       0   402.6    .045       0   417.1      .1       0
Bank Sta=402.6,417.1
XS Rating Curve= 0 ,0
Exp/Cntr=0.3,0.1

Type RM Length L Ch R = 1 ,11431   ,107.6,108.3,108.8
XS GIS Cut Line= 2
     2421405.363      556559.996     2421826.907      555840.219
#Sta/Elev= 30
       0 2578.24    33.9 2579.23    75.6 2576.76    96.9 2573.23   135.9 2564.15
   188.6 2557.11   200.8 2553.55     236 2537.46   269.4 2525.94   307.4 2508.47
   330.7 2498.91   344.5 2496.53   376.9 2496.74   399.42492.183   406.7 2491.43
   412.6 2492.27   418.6 2494.37   432.5  2495.4   446.4 2498.76   469.6 2500.69
     516 2507.23   534.5 2510.99   567.5 2519.31   673.6 2536.51   696.7 2541.93
   752.4 2552.94   766.3 2556.91   780.9 2562.64     808 2571.31   834.1 2580.93
#Mann= 3 ,-1 , 0
       0      .1       0   399.4    .045       0   412.6      .1       0
#XS Ineff= 2 , 0
          373.54 2497.04
Permanent Ineff=
       F       F
Bank Sta=399.4,412.6
XS Rating Curve= 0 ,0
Exp/Cntr=0.3,0.1

Type RM Length L Ch R = 1 ,11323   ,162.5,163.3,163.8
XS GIS Cut Line= 3
     2421479.659      556597.788     2421711.787      556242.311
     2421937.182      555901.841
#Sta/Elev= 30
       0 2557.34    22.8  2554.8    56.2 2553.46     133 2557.09   170.1 2550.98
   204.3 2546.52     233 2540.19   251.5 2533.68   265.2 2526.98   299.8 2507.81
     331 2494.88   338.1 2493.79   357.2 2494.21   369.9 2492.08   417.12489.746
   424.6 2489.06   430.6 2489.91   440.6 2493.96   476.8    2495   510.4 2498.44
   527.5 2501.28   596.7 2518.54   639.9  2532.6   665.2  2538.8   694.2  2548.4
   732.2 2563.21   759.8 2572.38   793.4 2585.96   807.8 2590.57   832.9 2603.45
#Mann= 3 ,-1 , 0
       0      .1       0   417.1    .045       0   430.6      .1       0
Bank Sta=417.1,430.6
XS Rating Curve= 0 ,0
Exp/Cntr=0.3,0.1

Type RM Length L Ch R = 1 ,11160   ,162.7,163.1,162.3
XS GIS Cut Line= 2
 2421586.3039554556663.5643085572422079.30570069 555986.20928807
#Sta/Elev= 30
       0 2555.98    35.7 2551.81    99.6 2543.05   122.5 2539.26   139.9  2535.1
   169.3 2529.37   182.7 2525.73   194.3 2523.94   235.1 2515.15   268.6 2506.23
   289.4  2499.5   311.5  2493.6     371  2486.8   406.7 2486.78   436.4 2484.97
   445.8 2484.12   448.72484.831   456.2 2489.18   485.9 2491.22   506.9 2498.69
   580.6 2511.13   623.6 2524.52     659 2533.14     684 2540.88   703.5 2549.73
   715.2 2556.11     761 2584.77   799.2 2610.57   826.4 2630.38   837.8 2640.12
#Mann= 3 ,-1 , 0
       0      .1       0   436.4    .045       0   448.7      .1       0
Bank Sta=436.4,448.7
XS Rating Curve= 0 ,0
Exp/Cntr=0.3,0.1

Type RM Length L Ch R = 1 ,10997   ,129.7,130.7,130.7
XS GIS Cut Line= 2
2421697.22044235556742.0090743292422205.43849257556083.700801124
#Sta/Elev= 30
       0 2556.91    59.8 2552.33   158.8 2542.03   247.2 2526.27   261.9 2522.17
   280.5 2514.93   306.7 2502.99   326.3 2491.38   342.7 2489.98   355.5  2484.2
   362.9 2482.16   390.92480.034   398.3 2479.69   405.8 2480.02   421.1  2482.6
   458.2 2483.48   469.6 2485.57   495.2 2494.54   512.4  2496.6   529.5 2500.92
   581.5 2520.22   629.3 2534.39   652.1 2542.56   681.3  2556.5   706.3 2570.63
   740.5 2592.72   782.3 2622.25   807.6 2641.81   822.7    2656   831.7  2662.4
#Mann= 3 ,-1 , 0
       0      .1       0   390.9    .045       0   405.8      .1       0
Bank Sta=390.9,405.8
XS Rating Curve= 0 ,0
Exp/Cntr=0.3,0.1

Type RM Length L Ch R = 1 ,10866   ,148.2,151.6,153.9
XS GIS Cut Line= 2
     2421771.371         556808.2422337.08761149556166.292198876
#Sta/Elev= 30
       0 2555.98    69.8  2548.4   104.7 2542.79   165.2 2527.71   245.5 2510.38
     311  2487.9   324.9 2487.11   367.4  2477.8   381.5 2478.22     391 2477.15
   407.1 2477.94   418.72476.324   426.9 2475.33   431.3 2476.25   443.4 2478.76
   465.6 2479.12   492.1 2486.87   509.9 2495.76   524.3  2498.4   537.4  2507.4
   574.2 2525.42   625.6 2543.33   645.1 2551.65   673.6 2565.77   697.4 2580.08
   718.8 2593.94   741.4 2610.48   789.6  2639.1   812.3  2650.7   855.5 2670.11
#Mann= 3 ,-1 , 0
       0      .1       0   418.7    .045       0   431.3      .1       0
Bank Sta=418.7,431.3
XS Rating Curve= 0 ,0
Exp/Cntr=0.3,0.1

Type RM Length L Ch R = 1 ,10714   ,137.2,136.3,135.5
XS GIS Cut Line= 3
      2421798.91      556841.7852422226.24737755556551.144774571
2422431.52058738556280.642821612
#Sta/Elev= 30
       0 2553.59    46.7 2545.82    98.8 2533.54   185.9 2515.93   205.2 2509.84
   247.3 2489.57   268.3  2483.6     302 2481.25   335.8 2481.51   346.1 2480.02
   363.3 2473.59   389.2 2474.32   406.5 2471.42   412.3 2470.77   418.62471.634
   442.2 2475.06   504.4 2477.51   527.4 2483.08   540.5 2489.95   550.2 2496.74
   561.6 2500.18   578.7  2512.3   639.8 2545.04   679.5 2573.71   688.1 2584.69
   692.7 2589.03   728.2 2613.16   778.5 2628.85   809.9 2637.13   856.4  2645.3
#Mann= 3 ,-1 , 0
       0      .1       0   406.5    .045       0   418.6      .1       0
Bank Sta=406.5,418.6
XS Rating Curve= 0 ,0
Exp/Cntr=0.3,0.1

Type RM Length L Ch R = 1 ,10578   ,172.6,171.9,171.4
XS GIS Cut Line= 3
     2421888.009      556974.8752422339.79709311556626.844584939
2422462.09835878556389.145005622
#Sta/Elev= 30
       0 2544.27    49.1 2532.89      69 2531.06    86.6 2526.64   191.7 2510.22
   203.1 2506.41   253.2 2482.64   268.3 2477.16   303.7 2476.29   349.1 2478.42
   357.1 2477.23   373.9 2469.76   402.4 2467.89   409.7 2467.22   417.42467.749
   515.7 2472.49   550.9    2479   568.1 2484.19   588.8 2494.86   600.7 2497.45
   606.4 2500.16   615.4 2507.41   637.9 2521.72   651.4 2536.03   668.1  2548.3
   691.9 2564.89   710.6 2575.58   741.4 2590.43   784.8 2606.43   837.6 2619.71
#Mann= 3 ,-1 , 0
       0      .1       0   402.4    .045       0   417.4      .1       0
Bank Sta=402.4,417.4
XS Rating Curve= 0 ,0
Exp/Cntr=0.3,0.1

Type RM Length L Ch R = 1 ,10406   ,156.3,154.7,154.9
XS GIS Cut Line= 3
     2422000.413      557136.3092422446.92512817556741.699115303
2422558.38232342556498.485646846
#Sta/Elev= 30
       0 2545.72    26.9 2539.25    85.7 2527.18   120.3  2517.1   134.5 2516.08
   171.1 2510.55   207.9  2503.1   219.5 2499.03   267.1 2474.55   272.5 2472.89
   325.8 2469.16   352.5 2465.77   389.5 2464.19   398.12462.527   405.9 2462.05
   411.2 2462.58   419.2 2463.84   434.8 2464.34   475.3 2464.16   503.8 2471.37
   556.7 2478.14   599.4 2488.81   616.8 2491.25   663.7 2516.04   687.2 2529.84
   704.8 2541.85     740 2557.59   775.2 2566.94   822.6  2575.1   863.4 2584.84
#Mann= 3 ,-1 , 0
       0      .1       0   398.1    .045       0   411.2      .1       0
Bank Sta=398.1,411.2
XS Rating Curve= 0 ,0
Exp/Cntr=0.3,0.1

Type RM Length L Ch R = 1 ,10251   ,209.5,212.7,212.6
XS GIS Cut Line= 3
     2422105.911      557221.9422422538.57903898556830.757035353
     2422666.161      556575.703
#Sta/Elev= 30
       0 2540.16    97.7 2521.58   134.5 2512.41   159.9  2504.1   176.2  2501.5
   240.9 2478.45   251.6 2473.11   267.3 2470.55   285.2 2464.26   316.3 2460.91
   363.9  2461.5   380.6 2458.63   406.3  2460.3   448.8 2459.04   457.3 2458.26
     463 2459.05   478.1 2468.75   548.2 2475.06   573.4 2481.57   587.8 2482.75
   610.2 2495.33   641.5 2506.19   650.6  2510.9   680.2 2520.34   699.6 2525.15
   766.5  2538.3   802.2 2548.85   829.2 2554.94     838 2554.82   868.5  2558.2
#Mann= 3 ,-1 , 0
       0      .1       0   448.8    .045       0     463      .1       0
Bank Sta=448.8,463
XS Rating Curve= 0 ,0
Exp/Cntr=0.3,0.1

Type RM Length L Ch R = 1 ,10039   ,89,92.3,94.9
XS GIS Cut Line= 3
2422183.62017477557279.2084833232422412.88656519557172.405287249
2422867.97510968556765.192249094
#Sta/Elev= 30
       0 2531.22    18.7 2530.26      54 2532.43    91.5 2525.15   121.6 2516.05
   186.4 2491.85   199.8 2489.03   234.9 2484.93   247.6 2480.37   259.6 2478.99
   279.3 2469.14   309.5 2457.07   409.7 2454.85   435.2 2452.86   443.7 2452.22
   449.4 2452.95   471.5    2457   501.5 2459.81   513.5 2463.88     553 2470.34
   568.3 2476.22   579.5 2478.39   591.4 2487.02   627.4 2496.99   699.4 2506.81
   724.1 2514.89   759.4 2517.63   780.8 2521.95  851.712532.321   863.6 2534.13
#Mann= 4 ,-1 , 0
       0      .1       0   435.2    .045       0   449.4      .1       0
  851.71     .05       0
Bank Sta=435.2,449.4
XS Rating Curve= 0 ,0
Exp/Cntr=0.3,0.1

Type RM Length L Ch R = 1 ,9947    ,107.2,102.7,96.5
XS GIS Cut Line= 5
2422493.75712941557619.688867278  2422488.490165557251.001357976
2422552.43539806557143.9850892762422635.96516872557101.770699449
2422904.58035407  556805.0650372
#Sta/Elev= 30
       0 2569.33    28.8 2565.16    56.8 2556.71    84.8 2550.49   128.8 2537.25
   168.8 2521.87   212.8 2511.29   232.8  2503.8   281.8 2481.51   320.8 2468.14
   348.8 2465.86   380.9 2471.87   392.2  2470.4   419.9  2460.9   434.6 2457.63
   555.82450.232   563.2 2449.36     5692450.034     609 2451.67   644.8 2457.34
   682.6 2471.12   693.4  2476.5   707.1 2478.95   725.8 2485.97   760.9 2492.08
   792.1  2494.4   847.4 2515.28   860.7 2518.95     913 2526.91   987.2    2534
#Mann= 3 , 0 , 0
       0      .1       0   555.8    .045       0     569      .1       0
Bank Sta=555.8,569
XS Rating Curve= 0 ,0
Exp/Cntr(USF)=0,0
Exp/Cntr=0.3,0.1

Type RM Length L Ch R = 1 ,9844    ,128.5,125.8,122.3
XS GIS Cut Line= 3
2422548.47171193557641.7462137412422546.98962274557333.692715553
     2422924.084      556837.033
#Sta/Elev= 30
       0 2553.89    27.2 2548.73   139.1 2533.06   195.1 2520.85     226 2510.55
   291.1 2479.09   303.1 2471.62   316.9  2470.6   331.3 2465.46     357 2461.35
   445.5 2454.92   448.4 2454.24   456.9 2447.71   462.6 2447.28   470.72447.847
   505.5 2450.05     558 2450.11   598.1 2453.32   623.3 2461.76   648.4 2473.23
   661.2 2475.79   674.4 2482.91   688.1 2484.33   700.9 2489.41   753.8 2497.21
  770.282501.602   839.4 2523.04   869.3 2529.38  896.512532.461   931.7 2534.67
#Mann= 5 ,-1 , 0
       0      .1       0   456.9    .045       0   470.7      .1       0
  770.28      .1       0  896.51      .1       0
#XS Ineff= 2 , 0
                          529.67         2453.48
Permanent Ineff=
       F       F
Bank Sta=456.9,470.7
XS Rating Curve= 0 ,0
Exp/Cntr=0.3,0.1

Type RM Length L Ch R = 1 ,9718    ,115.1,115.6,116.6
XS GIS Cut Line= 3
2422592.07379856 557637.245415342422802.75237531 557133.37248596
2422976.56220112556882.313848673
#Sta/Elev= 30
       0 2552.03    54.9 2544.87   115.6 2534.01   146.1 2524.15   218.9 2492.21
   240.8 2483.66   271.6 2473.18     289 2470.85   310.7  2464.9     341 2453.78
   354.2 2449.97     367 2448.22   384.4 2448.08   424.2 2442.34     432 2441.52
   438.8 2442.52   445.6  2444.7   460.9 2446.85   492.7 2447.13   522.1  2451.9
   540.5 2458.06   555.1 2463.84   563.3  2468.1   592.5 2471.34   598.4 2474.28
   617.6 2481.01   671.1 2495.27   690.5 2501.76   802.4 2531.08   851.5 2540.32
#Mann= 3 , 0 , 0
       0      .1       0   424.2    .045       0   438.8      .1       0
#XS Ineff= 2 , 0
                          469.22         2447.78
Permanent Ineff=
       F       F
Bank Sta=424.2,438.8
XS Rating Curve= 0 ,0
Exp/Cntr(USF)=0,0
Exp/Cntr=0.3,0.1

Type RM Length L Ch R = 1 ,9602    ,222.1,222.4,222.8
XS GIS Cut Line= 3
     2422705.125      557645.7992422782.24943302557417.777086374
2423052.60367096556903.223765771
#Sta/Elev= 30
       0  2550.8    45.6  2540.3    75.2 2531.62   117.4 2512.54   147.9 2500.19
   180.7 2488.77     223 2476.94   235.6 2470.48   250.7 2468.04   275.9 2456.88
   307.5  2444.8   331.6 2442.59   388.9 2443.43   397.9 2439.83   402.4 2439.17
     425  2440.1   428.4 2439.36     434 2437.99   440.2 2439.61   470.2 2447.78
   479.2 2449.22   506.3 2461.22   524.4 2463.06  533.372468.784     576 2482.58
   599.22488.637   646.4 2497.92   673.5 2504.58   727.7 2521.77     822 2546.78
#Mann= 5 ,-1 , 0
       0      .1       0   428.4    .045       0   440.2      .1       0
  533.37      .1       0   599.2      .1       0
#XS Ineff= 2 , 0
          375.55 2443.95
Permanent Ineff=
       F       F
Bank Sta=428.4,440.2
XS Rating Curve= 0 ,0
Exp/Cntr=0.3,0.1

Type RM Length L Ch R = 1 ,9380    ,179.8,177.1,173.8
XS GIS Cut Line= 4
2422902.98161149 557759.126552032422978.64902049557503.817730418
2423112.45722652557268.9878039262423176.13852792556983.808109681
#Sta/Elev= 30
       0 2550.66    67.3 2521.83    88.5 2513.92   146.5  2497.7   250.9 2466.56
   263.4 2461.49   276.9 2460.38   294.9 2453.29   326.6 2443.27   345.9 2435.43
   355.1 2434.04     369 2433.57   382.8 2435.28   394.6 2434.97   399.3 2434.11
  405.61 2431.21   410.4 2430.45   417.72431.167   433.4  2435.4   482.6 2433.28
   511.7 2436.57   555.4 2438.81  580.882441.174   597.7 2445.99   629.1  2458.7
   665.9 2469.93   699.4 2482.28   752.1 2504.94   796.5 2522.74   828.8 2533.42
#Mann= 4 ,-1 , 0
       0      .1       0  405.61    .045       0   417.7      .1       0
  580.88      .1       0
Bank Sta=405.61,417.7
XS Rating Curve= 0 ,0
Exp/Cntr=0.3,0.1

Type RM Length L Ch R = 1 ,9203    ,174.5,174.8,175.9
XS GIS Cut Line= 2
2423118.52238289557826.1261691442423317.14038289557029.867169144
#Sta/Elev= 30
       0 2515.53    36.6 2507.54      54 2502.35    90.2 2494.05   143.8 2478.92
   230.4 2456.74   267.5 2448.65   279.8 2444.73   300.5 2441.71   341.7 2427.58
   382.9 2427.29   396.72425.956   403.7 2425.36   408.6    2426   416.9 2429.17
  431.49 2429.32   449.9 2428.92   470.8 2429.88   514.8 2429.11     539 2431.88
   578.6 2434.46     589 2436.14   605.5 2441.12  643.132455.591   671.4 2468.69
   704.4 2480.79   741.5 2493.33   782.7 2505.97   807.5 2504.77   820.7 2505.94
#Mann= 5 ,-1 , 0
       0      .1       0   396.7    .045       0   408.6      .1       0
  431.49      .1       0  643.13      .1       0
Bank Sta=396.7,408.6
XS Rating Curve= 0 ,0
Exp/Cntr=0.3,0.1

Type RM Length L Ch R = 1 ,9028    ,211.3,211.2,210.8
XS GIS Cut Line= 2
2423270.30838289557860.1838457222423501.16538289557069.674845721
#Sta/Elev= 30
       0 2491.58    89.2 2474.01   135.3 2467.92   189.2 2457.87   289.2 2433.51
   305.8 2430.17   314.2 2427.37   326.7 2426.53   343.3 2423.76   372.5 2424.32
   393.2 2423.35   402.9 2420.99   405.8 2420.41   418.3    2421   435.2 2422.73
   472.5 2423.43  502.072425.776     535  2429.9   547.5 2432.27   555.8 2432.78
   596.4 2443.13   612.5  2448.2   631.9 2451.98   643.3 2456.45     660 2461.14
  699.472476.655   728.6 2485.79   763.9 2495.02   801.7 2506.78   823.5 2512.42
#Mann= 5 ,-1 , 0
       0      .1       0   402.9    .045       0   418.3      .1       0
  502.07      .1       0  699.47      .1       0
Bank Sta=402.9,418.3
XS Rating Curve= 0 ,0
Exp/Cntr=0.3,0.1

Type RM Length L Ch R = 1 ,8817    ,241,238.4,234.8
XS GIS Cut Line= 3
2423460.12672117557907.8720297312423625.92767658557382.888408995
2423658.68696102 557111.09281599
#Sta/Elev= 30
       0 2477.43    84.2  2472.8   135.6 2465.49   173.3  2455.1   253.1 2429.34
   261.4 2427.82   307.6 2423.21   314.2 2421.41   324.3 2416.85   328.5 2416.06
   341.1 2415.12   357.9 2416.72   383.1 2416.83   416.6 2415.77   439.3 2413.85
     446 2413.34   450.2 2413.79   466.9 2417.59  483.642419.025  490.332419.106
   508.9 2419.55   525.7 2422.97   538.2 2423.75   542.4 2425.14   599.2 2452.05
   623.3 2461.47   643.5 2467.41   707.9 2490.77   776.4  2510.3   824.3 2521.98
#Mann= 5 ,-1 , 0
       0      .1       0   439.3    .045       0   450.2      .1       0
  483.64      .1       0  490.33      .1       0
Bank Sta=439.3,450.2
XS Rating Curve= 0 ,0
Exp/Cntr=0.3,0.1

Type RM Length L Ch R = 1 ,8578    ,174.6,174.1,173.2
XS GIS Cut Line= 2
2423777.17635315557916.2702490942423812.16284572557133.483676577
#Sta/Elev= 30
       0 2431.13      11 2430.54    29.7 2433.78    45.7 2434.72  102.242431.674
   185.9 2426.37   233.1 2422.34   241.9 2420.82     274 2411.42  301.212408.701
     358 2408.38   374.72406.927     382 2405.72     386 2405.92   388.72407.158
   394.1 2409.68   398.1  2410.3   434.1 2412.68   442.1 2412.34   466.1 2416.56
   478.1 2416.88   486.1 2420.34   518.3 2429.91   533.6 2436.81   582.2 2461.62
   602.2 2470.36   642.3 2484.73   710.8 2505.91   770.4 2516.43   783.6 2517.85
#Mann= 5 ,-1 , 0
       0      .1       0  102.24     .05       0  301.21      .1       0
   374.7    .045       0   388.7      .1       0
#XS Ineff= 2 , 0
          322.96 2409.26
Permanent Ineff=
       F       F
Bank Sta=374.7,388.7
XS Rating Curve= 0 ,0
Exp/Cntr=0.3,0.1

Type RM Length L Ch R = 1 ,8404    ,133.3,138.4,142.5
XS GIS Cut Line= 3
2423866.66985835557888.5865506422423958.06181322 557664.30903585
2423948.61464515557128.636248248
#Sta/Elev= 30
       0 2426.03    10.8 2425.07   28.532426.943    58.3 2426.98   127.4  2424.3
  214.822418.424   247.9 2414.87   271.9  2406.8   279.9 2405.01   315.9 2405.03
   335.9 2403.16   348.1 2403.27   363.9 2401.37   371.9 2400.83   376.6 2401.42
   383.9 2403.25   419.9 2404.62   443.9 2409.16   451.9 2411.47   463.9 2412.58
   475.9 2420.18     501    2432   536.4 2446.28   559.9 2457.81   579.9 2465.75
   612.8 2473.86   635.9 2481.24   691.9 2496.14   739.9 2504.45   777.9 2508.59
#Mann= 5 ,-1 , 0
       0      .1       0   28.53     .05       0  214.82      .1       0
   363.9    .045       0   376.6      .1       0
#XS Ineff= 2 , 0
          313.63 2409.43  405.44         2409.66
Permanent Ineff=
       F       F
Bank Sta=363.9,376.6
XS Rating Curve= 0 ,0
Exp/Cntr=0.3,0.1

Type RM Length L Ch R = 1 ,8266    ,175.5,167.5,162.1
XS GIS Cut Line= 3
2423969.97475175557861.7750925812424097.27985528557551.194376679
2424017.27138289557132.205187938
#Sta/Elev= 30
       0 2419.16    76.9 2415.42   132.9 2414.33     172 2414.44  202.662412.893
  205.222412.417   234.2 2404.32   249.8 2403.25   262.8 2403.22   280.2 2401.04
   295.6 2397.86   301.7 2397.09     306 2397.76  316.592397.702   327.7 2398.75
   381.1 2399.77   409.6 2401.36   429.9 2403.39   449.8 2407.49   462.5 2407.75
   470.6  2411.9   503.2 2425.06   519.5 2433.25   539.9 2441.93   588.7 2459.15
   613.1 2466.45   641.6 2472.46   682.3 2478.58   730.1 2487.77   762.2 2492.32
#Mann= 6 ,-1 , 0
       0     .05       0  202.66      .1       0  205.22     .05       0
   295.6    .045       0     306     .05       0  316.59      .1       0
#XS Ineff= 2 , 0
                          344.51            2404
Permanent Ineff=
       F       F
Bank Sta=295.6,306
XS Rating Curve= 0 ,0
Exp/Cntr=0.3,0.1

Type RM Length L Ch R = 1 ,8098    ,117.6,116.6,115.3
XS GIS Cut Line= 2
2424341.34097897557894.8581949482424081.34376577557096.154429176
#Sta/Elev= 30
       0 2471.43      55 2454.03   121.6 2434.49     198 2416.02   206.4 2414.75
   231.6 2407.03   290.5 2400.48   324.2 2398.64   345.2 2394.43   353.2 2395.22
  365.43 2394.24   383.1 2396.46   400.8 2396.72     423 2393.03   429.3 2392.16
   435.7 2392.91   446.2 2396.49     458 2396.31   467.2 2398.76     484 2400.04
     505  2404.9   515.1  2405.8   517.7 2406.67   526.1 2413.44   559.5 2432.62
   576.5 2439.91   603.9 2448.38   645.2  2457.1   715.4 2473.66     840 2497.11
#Mann= 4 ,-1 , 0
       0     .05       0  365.43      .1       0     423    .045       0
   435.7      .1       0
Bank Sta=423,435.7
XS Rating Curve= 0 ,0
Exp/Cntr=0.3,0.1

Type RM Length L Ch R = 1 ,7982    ,106,106.6,108.5
XS GIS Cut Line= 3
2424397.05023423557876.8383828862424401.81932228557638.205652964
2424149.96407433557063.521368867
#Sta/Elev= 30
       0 2469.43    34.3 2458.16    74.3 2443.59   134.3 2424.81   238.3 2399.63
   268.8 2398.12   299.4 2393.14   316.9 2393.11   325.6 2391.48   359.1 2391.51
   404.2 2393.52   417.3 2392.71     426 2393.23   442.9  2392.4   448.12390.171
   456.6 2389.36   463.32390.328   481.5 2396.46   500.3 2401.22   513.4 2408.04
   526.5 2408.07   530.8 2409.41   539.6 2414.92   570.1  2429.4   587.6 2436.92
   596.3 2439.74     619 2444.91   679.8 2455.77   757.9 2475.89   866.1 2494.96
#Mann= 4 ,-1 , 0
       0     .05       0   359.1      .1       0   448.1    .045       0
   463.3      .1       0
#XS Ineff= 2 , 0
          314.96 2395.12
Permanent Ineff=
       F       F
Bank Sta=448.1,463.3
XS Rating Curve= 0 ,0
Exp/Cntr=0.3,0.1

Type RM Length L Ch R = 1 ,7875    ,214,218.7,220.6
XS GIS Cut Line= 4
     2424490.829      557837.984 2424494.5853969 557625.78761989
2424381.51669115557338.0167497792424414.90016969557022.768684433
#Sta/Elev= 30
       0 2460.64    39.4 2444.49    91.4 2426.78   199.4 2395.77   224.3  2392.3
   301.6 2390.48   314.5 2387.74  333.532390.347   344.6 2390.51   361.8 2388.55
   395.4 2389.23   407.7 2387.03   413.9  2386.1   419.2 2386.91   426.2 2389.06
  433.482389.285     452 2389.94   456.3 2391.72   473.5 2403.41     495 2411.91
   506.4 2415.23   518.8    2416     565 2433.81     621 2448.98   645.5 2454.76
   697.8 2463.48   712.5 2468.09     734  2472.8   767.1 2477.91   838.4  2492.3
#Mann= 5 ,-1 , 0
       0     .05       0  333.53      .1       0   407.7    .045       0
   419.2      .1       0  433.48      .1       0
#XS Ineff= 2 , 0
          290.49 2391.93
Permanent Ineff=
       F       F
Bank Sta=407.7,419.2
XS Rating Curve= 0 ,0
Exp/Cntr=0.3,0.1

Type RM Length L Ch R = 1 ,7656    ,151.9,152.7,153.8
XS GIS Cut Line= 2
2424616.10246422557831.0348120622424558.79928753557022.703134638
#Sta/Elev= 30
       0 2462.76    36.5 2447.06   112.7  2417.5   144.8 2405.68   166.6 2399.69
     217 2390.56   249.1 2386.84  341.03 2385.72   381.4 2383.81   392.32380.281
   393.4 2380.13   405.32380.296   413.5 2381.76  438.892383.821   445.8 2384.71
     457 2388.82   473.6 2399.66   493.6 2411.15   509.7 2418.14   517.7  2423.9
   525.7 2427.18   565.8 2431.48   569.8 2433.17   573.8  2437.1   577.8 2439.48
     663 2461.49   694.1 2471.51   754.3 2486.36   762.3 2486.66   810.4 2500.43
#Mann= 5 ,-1 , 0
       0     .05       0  341.03      .1       0   392.3    .045       0
   405.3      .1       0  438.89      .1       0
Bank Sta=392.3,405.3
XS Rating Curve= 0 ,0
Exp/Cntr=0.3,0.1

Type RM Length L Ch R = 1 ,7504    ,144.2,143.6,143.3
XS GIS Cut Line= 3
     2424720.105      557821.6452424735.78802103557364.441549795
     2424679.621      556991.716
#Sta/Elev= 30
       0 2474.28   111.1 2420.43   143.1 2407.45   171.2 2397.97   195.2 2393.07
   255.2 2383.73   283.2 2380.99   323.2 2380.21   335.9 2378.82  352.782379.334
   407.3 2379.59   421.5 2376.52   427.3 2376.12     4332376.683   439.3 2380.09
  452.062392.468   463.4 2401.63   479.3 2407.64   515.9 2418.16   532.1 2420.11
   556.4 2429.45   572.6 2434.45   595.7 2438.39   641.3 2451.09   673.7 2458.59
   689.9 2463.94   742.4 2484.56   760.9 2490.36   806.6  2501.8   834.4 2507.21
#Mann= 5 ,-1 , 0
       0     .05       0  352.78      .1       0   421.5    .045       0
     433      .1       0  452.06      .1       0
Bank Sta=421.5,433
XS Rating Curve= 0 ,0
Exp/Cntr=0.3,0.1

Type RM Length L Ch R = 1 ,7360    ,103.9,103.6,103
XS GIS Cut Line= 4
2424951.14924401 557785.627113612424868.77983835557597.600390698
2424875.54808134  557381.71105332424767.90177701556989.156556805
#Sta/Elev= 30
       0 2500.14    20.8 2489.32     132 2426.94   186.7 2399.34   199.8 2393.23
   216.3 2386.68   236.3 2380.06   252.3 2377.28  355.83 2376.24   360.3 2375.55
     369 2372.67   372.3 2371.63   376.3  2371.5   383.82372.559   400.4 2376.76
   408.4 2381.97   416.4 2384.87   441.1 2390.73   474.2 2399.81     495 2402.15
   503.3  2406.9   520.8  2413.1  552.852421.183   586.2 2428.84   623.5 2439.42
   660.9  2451.3   686.8 2460.58   764.5 2483.68   786.7 2488.77   828.3 2496.38
#Mann= 5 ,-1 , 0
       0     .05       0  355.83      .1       0     369    .045       0
   383.8      .1       0  552.85      .1       0
Bank Sta=369,383.8
XS Rating Curve= 0 ,0
Exp/Cntr=0.3,0.1

Type RM Length L Ch R = 1 ,7257    ,131.8,132.3,132.4
XS GIS Cut Line= 4
 2425061.2453436557780.8004221672424976.09374576557583.098511317
 2424977.5439337557356.8691929752424839.65703227557007.856812062
#Sta/Elev= 30
       0 2523.73    37.3  2504.8    85.2 2477.24  168.852421.793   219.9 2390.27
   239.7 2379.67   251.7 2375.33   259.8 2374.25   295.8 2374.17   323.7  2372.9
   355.7 2373.54  367.332371.462   373.42369.726   379.7 2368.91  385.18 2369.67
   399.7 2378.04   403.7  2379.3   448.2 2386.89  466.422393.424     474 2395.29
   491.2 2395.38   510.2 2397.51   521.1 2403.95   524.3 2404.96   564.7  2414.3
   590.1 2422.23   640.9 2434.86   767.9 2470.88   804.1 2483.28   816.8 2486.56
#Mann= 6 ,-1 , 0
       0      .1       0  168.85     .05       0  367.33      .1       0
   373.4    .045       0  385.18      .1       0  466.42      .1       0
Bank Sta=373.4,385.18
XS Rating Curve= 0 ,0
Exp/Cntr=0.3,0.1
